HEC-RAS study OLDFLDFK1.prj: OLDFLDFK1

--- OLDFLDFK1.g01 (geometry) --- (continued)

Type RM Length L Ch R = 1 ,19591   ,422.6,424.2,426
XS GIS Cut Line= 2
2218793.01746333523840.3959944012219543.73261397524123.314763859
#Sta/Elev= 30
       0 2692.11    16.2 2687.09     106 2652.19   142.8 2635.34   204.3 2621.11
   272.7 2618.01   349.6 2618.75   353.9 2617.81   363.2 2612.26   375.6 2610.54
   400.9 2613.67   443.7 2610.38   452.2 2611.48   478.1 2610.37   490.7 2614.78
   502.9 2614.48   517.2 2609.45   525.4 2606.34   580.4 2606.34   587.2 2609.56
   606.1 2619.32   623.2 2620.53   631.7  2632.3   644.6 2641.77   687.3 2660.29
   700.1 2667.63     713 2669.98   755.7 2692.77   782.3 2700.68   802.3 2703.07
#Mann= 3 ,0,0
       0      .1       0   517.2    .045       0   587.2      .1       0
#XS Ineff= 2 , 0
          344.23 2625.03
Permanent Ineff=
       F       F
Bank Sta=517.2,587.2
XS Rating Curve= 0 ,0
Exp/Cntr(USF)=0,0
Exp/Cntr=0.3,0.1

Type RM Length L Ch R = 1 ,19167   ,438.4,437.9,438
XS GIS Cut Line= 2
2218671.16631015 524228.358861432219420.48087282524540.689978207
#Sta/Elev= 30
       0 2696.55    74.8  2671.1   109.4 2656.76   152.8 2635.47   204.8 2620.73
   248.1  2618.2   287.1 2613.38   417.4 2614.75   438.8 2611.62   457.1 2612.13
   495.1 2606.18     500 2603.86   509.1 2603.41   558.1 2603.48   564.5 2606.07
   577.5 2615.13   582.5 2616.88   590.5 2617.16   594.8 2619.15     604 2637.22
   607.8 2639.97   616.2 2642.64   629.5 2649.94   661.7 2660.19   694.5 2666.73
   733.5 2683.22   746.5 2690.84   761.1 2694.87   798.5 2700.73   811.8 2701.45
#Mann= 3 ,-1,0
       0      .1       0   495.1    .045       0   564.5      .1       0
#XS Ineff= 2 , 0
           406.2 2623.07
Permanent Ineff=
       F       F
Bank Sta=495.1,564.5
XS Rating Curve= 0 ,0
Exp/Cntr(USF)=0,0
Exp/Cntr=0.3,0.1

Type RM Length L Ch R = 1 ,18729   ,366.8,367.5,367.8
XS GIS Cut Line= 3
2218540.91162916524654.1376035842219128.62952465524891.551464257
 2219291.6267798 524890.83697011
#Sta/Elev= 30
       0 2723.83    23.3 2716.61    46.7 2705.32    72.5 2685.19    89.8 2674.37
   115.7 2655.42   154.5 2636.19   164.6 2629.62   189.7 2620.46   207.6 2609.56
   305.5  2611.5   382.8 2610.26   417.7 2608.87   430.6 2606.24   439.2 2606.31
   446.5 2603.57   452.2 2601.51   538.5 2601.48  548.12 2603.44     560 2611.21
   568.7 2613.64   594.8 2609.58   641.4 2615.38   645.4 2617.98   653.4 2626.91
   657.4 2629.12   685.4 2642.86   705.4 2650.56   749.4 2673.34   796.9 2688.76
#Mann= 3 ,-1,0
       0      .1       0   446.5    .045       0  548.12      .1       0
#XS Ineff= 2 , 0
          379.04 2615.83
Permanent Ineff=
       F       F
Bank Sta=446.5,548.12
XS Rating Curve= 0 ,0
Exp/Cntr(USF)=0,0
Exp/Cntr=0.3,0.1

Type RM Length L Ch R = 1 ,18361   ,396.7,395,392.9
XS GIS Cut Line= 3
2218494.69222623525028.0945909362218952.68449164525217.173966564
2219210.39267768525183.559855341
#Sta/Elev= 30
       0 2702.82    27.6 2697.22    79.5  2671.8    92.5 2667.85   118.4  2651.6
   131.4 2646.58   155.1 2633.42   164.3  2626.5   174.7 2613.65   183.4 2606.41
     202 2604.38   228.6 2607.98   269.9 2609.69   285.9 2604.81   326.2 2607.48
   354.2 2601.76   360.8 2599.59     417 2599.58   447.3 2599.58  454.522601.817
   464.6 2609.78     469  2611.1   536.7 2606.76     612  2609.2   660.4 2632.64
   671.2 2634.73   680.5 2639.73   704.7 2641.04   719.8 2649.22   755.4 2661.94
#Mann= 3 ,-1,0
       0      .1       0   354.2    .045       0  454.52      .1       0
#XS Ineff= 2 , 0
          262.76 2621.33  493.07         2622.04
Permanent Ineff=
       F       F
Bank Sta=354.2,454.52
XS Rating Curve= 0 ,0
Exp/Cntr(USF)=0,0
Exp/Cntr=0.3,0.1

Type RM Length L Ch R = 1 ,17967   ,346.6,340.4,332.6
XS GIS Cut Line= 2
2218399.45224443525423.0603978032219095.54446434525693.373875552
#Sta/Elev= 30
       0 2674.59    76.4 2663.89    90.9 2658.98   103.8 2657.42     151 2645.47
     166 2640.21   219.6 2628.81   245.4 2614.21   249.7 2608.05   253.9 2604.75
  269.78 2600.75   275.4 2598.01   282.1 2597.84   399.8 2597.85  404.52 2600.81
   408.4  2606.9   421.3 2608.27   441.1 2606.18   455.6 2607.29   477.1 2605.46
   567.2 2605.26   602.5 2603.05   644.4 2604.53   651.3 2607.11   665.9 2616.74
   679.1 2628.76   700.2 2645.13   721.7 2657.04   738.8 2670.22   746.7 2671.92
#Mann= 3 ,0,0
       0      .1       0  269.78    .045       0  404.52      .1       0
#XS Ineff= 2 , 0
                          418.25         2619.32
Permanent Ineff=
       F       F
Bank Sta=269.78,404.52
XS Rating Curve= 0 ,0
Exp/Cntr(USF)=0,0
Exp/Cntr=0.3,0.1

Type RM Length L Ch R = 1 ,17626   ,372.9,338.9,301.1
XS GIS Cut Line= 3
2218398.05165647525806.8215009282218756.60217618525909.064422564
2218963.88919538525967.889117204
#Sta/Elev= 30
       0 2641.41      23 2635.78    56.3 2630.06     104 2620.08   123.4 2614.27
   131.2 2611.02   139.5 2605.35   147.8 2598.38   151.9 2596.28   155.7 2596.25
   255.9 2596.31   264.3 2598.52   301.7  2602.9   326.6 2602.03   364.1 2603.66
   372.4 2604.95   409.8  2601.2   430.9 2601.42   447.2 2600.09     468 2601.99
   484.7 2602.03   508.6  2600.1   513.8 2602.16   517.9 2608.14   522.1  2618.1
   526.2 2622.75   534.5 2629.15   559.5 2641.07   576.1  2646.4   588.3 2648.62
#Mann= 3 ,-1,0
       0      .1       0   147.8    .045       0   264.3      .1       0
#XS Ineff= 2 , 0
                          373.86          2610.8
Permanent Ineff=
       F       F
Bank Sta=147.8,264.3
XS Rating Curve= 0 ,0
Exp/Cntr(USF)=0,0
Exp/Cntr=0.3,0.1

Type RM Length L Ch R = 1 ,17287   ,307.1,276.9,228.1
XS GIS Cut Line= 3
2218330.82343402526278.8196460132218839.23686626526106.547325997
 2218945.6815518526007.105580297
#Sta/Elev= 30
       0 2691.63    47.9 2666.18      56 2665.19    77.4 2655.79    85.9 2653.41
   123.9 2637.28   157.7 2624.52     220 2605.33   232.6 2594.45   237.9 2591.92
   242.1 2591.81   292.6 2591.97     302 2594.32   318.2 2597.28   339.9 2598.66
   368.9 2597.96   385.8 2601.87   457.6 2600.39   491.2 2598.63   507.1 2599.42
   533.6 2603.25     549 2601.41   563.9 2604.96   565.5 2606.15   570.9 2613.67
   576.4  2618.5   592.2 2624.91   644.3 2635.48     656 2636.11   682.5 2640.04
#Mann= 3 ,-1,0
       0      .1       0   232.6    .045       0     302      .1       0
#XS Ineff= 2 , 0
                           533.6            2610
Permanent Ineff=
       F       F
Bank Sta=232.6,302
XS Rating Curve= 0 ,0
Exp/Cntr(USF)=0,0
Exp/Cntr=0.3,0.1

Type RM Length L Ch R = 1 ,17010   ,376.8,357.4,337.5
XS GIS Cut Line= 4
2218696.63899571526517.8887373182218773.96423607526307.700467677
2218988.77064324526231.3050478632218995.07546594526074.456194501
#Sta/Elev= 30
       0 2646.89     9.5 2638.53    17.8 2633.21    73.2 2604.13    78.1 2600.98
    93.7 2593.34   97.38 2590.79     103    2589   141.4 2589.02   145.7 2589.31
   149.9 2590.83   165.3 2592.78   179.8  2593.5   209.6 2599.58     239 2599.18
   268.8 2597.69     290 2598.25   315.5 2596.66   332.4 2599.84   353.7 2601.67
   404.6 2601.69   430.1 2600.66   446.4 2602.04   466.1  2600.3   482.1 2603.75
   538.2 2605.03   550.2 2606.06   558.2 2607.44   590.2 2616.66   608.9 2618.94
#Mann= 3 ,-1,0
       0      .1       0   97.38    .045       0   149.9      .1       0
Bank Sta=97.38,149.9
XS Rating Curve= 0 ,0
Exp/Cntr(USF)=0,0
Exp/Cntr=0.3,0.1

Type RM Length L Ch R = 1 ,16653   ,330.7,309.7,293.8
XS GIS Cut Line= 3
 2219088.5415245526724.2066197142219075.93623279526277.419058046
2219091.34270043526050.523807293
#Sta/Elev= 30
       0 2724.45    18.9 2724.03      55 2717.45    71.1 2711.82    83.1 2704.89
   103.1 2688.84   138.6 2655.56   155.1 2645.31   159.1 2641.18   163.1 2635.44
   166.8 2624.93   171.1 2609.21   183.1 2596.49  195.45 2589.47   203.1 2585.95
   207.1  2585.7   267.1 2585.71   271.1    2586   277.1 2589.44   291.1 2596.02
   303.1  2599.2   343.2 2597.79   439.2 2599.59   450.5 2601.16   463.2 2599.68
   491.3  2599.5   523.4 2602.96   571.5 2603.25   651.7 2616.62   674.4 2621.55
#Mann= 3 ,0,0
       0      .1       0  195.45    .045       0   277.1      .1       0
#XS Ineff= 2 , 0
                          310.37         2614.17
Permanent Ineff=
       F       F
Bank Sta=195.45,277.1
XS Rating Curve= 0 ,0
Exp/Cntr(USF)=0,0
Exp/Cntr=0.3,0.1

Type RM Length L Ch R = 1 ,16343   ,245,242.6,240.5
XS GIS Cut Line= 2
2219461.09792388526628.9666379162219227.19973329525983.295584847
#Sta/Elev= 30
       0 2721.82    25.3 2719.31    50.5 2710.58    72.1 2697.46   106.1 2672.46
   127.4 2654.81   140.2 2646.13   144.4 2641.74   148.7 2635.34   152.9  2626.7
   157.2 2612.57   161.4 2600.52   174.2 2589.11   178.5 2585.76   182.7 2585.41
     255 2585.41   259.3  2585.7     266 2588.95   276.3 2591.45   297.6 2593.72
   309.7 2599.02   314.6 2599.51   357.1  2597.6   369.9 2598.61   382.7 2596.93
   531.6 2601.94   586.9  2609.8   628.3 2617.96   650.7 2624.09   686.7 2637.29
#Mann= 3 ,0,0
       0      .1       0   174.2    .045       0     266      .1       0
Bank Sta=174.2,266
XS Rating Curve= 0 ,0
Exp/Cntr(USF)=0,0
Exp/Cntr=0.3,0.1

Type RM Length L Ch R = 1 ,16101   ,213,211.8,211.6
XS GIS Cut Line= 3
2219710.40258212526577.1448831152219560.53966958526205.989071698
 2219477.9049795 525952.48264956
#Sta/Elev= 30
       0 2695.44     5.9 2695.39    17.2 2693.05    25.8 2693.45    34.5 2690.84
    43.1 2689.97    86.2 2670.17   130.8 2655.55   142.3 2650.78   164.6 2638.78
   168.2 2636.38   176.8 2628.28   187.6 2620.92   191.3 2616.51   198.4 2603.79
     207 2592.64   211.3 2588.08   215.7 2585.25   219.6 2585.16   306.2 2585.16
   310.6 2585.46   314.3 2588.29   323.5 2591.25   349.4 2594.25   379.7  2593.6
   405.3 2596.08   430.6 2595.72   619.9 2601.86   649.3 2609.53   666.9 2610.19
#Mann= 3 ,0,0
       0      .1       0   211.3    .045       0   314.3      .1       0
Bank Sta=211.3,314.3
XS Rating Curve= 0 ,0
Exp/Cntr(USF)=0,0
Exp/Cntr=0.3,0.1

Type RM Length L Ch R = 1 ,15889   ,221.1,237.3,250.2
XS GIS Cut Line= 4
2219816.84726766 526574.343707182219868.66902246526402.071387163
2219753.82080912526120.5532056732219758.02257302525869.847959471
#Sta/Elev= 30
       0 2676.11     9.6 2674.28    26.3 2668.45    51.3 2658.14    77.5  2650.4
   105.6 2638.51   118.2 2634.57   134.9 2625.84   154.5 2612.61   180.6 2599.93
   198.1 2596.44   228.4 2597.85   254.6  2597.4   258.6 2596.48   268.2 2586.34
   271.6 2584.24   375.3 2584.29   382.4 2584.65   386.5 2586.53   392.5 2588.39
   422.8 2589.39   447.9 2592.45     466 2592.02   483.9 2594.57   559.3 2589.39
   583.3 2596.08   627.4 2612.87   707.3 2649.64   715.3 2651.31   734.7 2662.86
#Mann= 3 ,-1,0
       0      .1       0   268.2    .045       0   386.5      .1       0
#XS Ineff= 2 , 0
                          483.15         2603.74
Permanent Ineff=
       F       F
Bank Sta=268.2,386.5
XS Rating Curve= 0 ,0
Exp/Cntr(USF)=0,0
Exp/Cntr=0.3,0.1

Type RM Length L Ch R = 1 ,15651   ,219.1,301,370.7
XS GIS Cut Line= 5
2219867.26843449 526579.946059052219984.91782377526437.086086354
2220054.94722215526281.6208219492220011.52899516526070.132038839
2220066.15192589525907.663834596
#Sta/Elev= 30
       0 2662.87    20.3 2658.57    45.5 2649.49   107.8 2620.79     139 2600.37
   161.7 2591.79   189.4 2594.15   360.1 2597.19   364.2 2596.61   368.3  2594.2
   378.3 2585.36   384.6 2582.45   507.1 2582.53  512.45 2585.35   523.4 2589.31
   531.6 2589.52   543.9 2587.62     552 2590.56   568.4 2593.06   576.7 2593.03
   585.4 2589.69   593.6 2591.51   623.3 2612.55   639.1 2629.65   652.7 2640.71
   670.6 2648.94   682.2 2656.77   692.8 2661.01   724.5 2682.71   742.9 2692.84
#Mann= 3 ,0,0
       0      .1       0   378.3    .045       0  512.45      .1       0
#XS Ineff= 2 , 0
           351.1 2604.27  572.85         2599.75
Permanent Ineff=
       F       F
Bank Sta=378.3,512.45
XS Rating Curve= 0 ,0
Exp/Cntr(USF)=0,0
Exp/Cntr=0.3,0.1

Type RM Length L Ch R = 1 ,15350   ,284.8,352.8,412.6
XS GIS Cut Line= 2
2219872.77801406526588.419755689  2220384.013405526231.765557637
#Sta/Elev= 30
       0 2658.89    16.3 2655.67    42.1  2647.4    79.5 2631.27    89.6 2628.56
   111.4  2617.1   117.5 2614.75   131.2 2604.38   154.2 2591.79   178.1 2589.21
   194.4 2584.24   379.7 2588.25   404.1 2587.53     448  2583.2   462.6 2584.34
   468.4 2582.98   474.1 2581.44     519 2581.52     524 2582.93     530 2586.08
     537 2586.58   550.4 2591.22     565 2594.34   574.8 2603.59   585.1 2609.71
   593.7 2613.29   599.9 2618.67   608.9  2620.6   618.7 2630.52   623.3 2632.17
#Mann= 3 ,-1,0
       0      .1       0   468.4    .045       0     524      .1       0
Bank Sta=468.4,524
XS Rating Curve= 0 ,0
Exp/Cntr(USF)=0,0
Exp/Cntr=0.3,0.1

Type RM Length L Ch R = 1 ,14998   ,263.5,275.5,284.7
XS GIS Cut Line= 3
2219877.43407409526594.938239727 2220123.2740435526520.441279298
2220376.56370896 526758.83155267
#Sta/Elev= 30
       0 2655.63    22.9 2649.54   115.9 2616.35   124.1 2610.54   132.4 2602.19
   141.5 2590.61   149.2 2585.15   157.5 2582.78   174.2 2581.19   211.8 2581.76
   266.5  2583.6   280.1 2585.34   297.7 2583.03   340.5 2582.47   362.5 2580.13
     379 2581.19   382.5 2580.24   386.4  2579.2   409.7 2579.11   450.6 2579.13
   456.4 2580.11   461.8 2583.79   473.9 2589.01   488.8 2587.26   515.5  2588.5
   532.3 2602.68   549.2 2612.39   560.2 2616.56   586.3 2623.22   604.7 2630.57
#Mann= 3 ,-1,0
       0      .1       0   382.5    .045       0   456.4      .1       0
Bank Sta=382.5,456.4
XS Rating Curve= 0 ,0
Exp/Cntr(USF)=0,0
Exp/Cntr=0.3,0.1

Type RM Length L Ch R = 1 ,14722   ,262.5,261.2,261.9
XS GIS Cut Line= 2
2219893.87960588526610.7589943372220166.99425956527001.523037301
#Sta/Elev= 30
       0 2647.38    49.3 2628.42    75.2 2616.52    95.3 2604.91   100.6 2600.78
   115.7 2581.46   121.2 2580.18   144.5 2578.87   168.9 2579.06   175.7 2577.76
   183.5 2575.18     193 2575.13   253.3 2575.23   256.7 2575.64     259 2577.56
   261.9 2579.76   266.5 2580.58   276.3 2580.56   290.6  2578.8   313.6 2581.25
   359.6 2580.36   382.6 2585.08   399.8 2584.97   412.9 2590.65   422.8 2592.72
   450.9 2610.92   454.4 2615.46   457.9 2622.23   461.7 2626.82   476.7 2637.27
#Mann= 3 ,-1,0
       0      .1       0   175.7    .045       0     259      .1       0
Bank Sta=175.7,259
XS Rating Curve= 0 ,0
Exp/Cntr(USF)=0,0
Exp/Cntr=0.3,0.1

Type RM Length L Ch R = 1 ,14461   ,246.4,220.1,197.7
XS GIS Cut Line= 2
2219652.97186099526718.0890091822219996.56824082527207.453550152
#Sta/Elev= 30
       0 2670.96    13.6 2665.91    28.2  2657.3    40.4 2652.35    52.7 2644.03
    62.4 2642.86    86.9  2627.9    96.4 2626.63   130.9 2609.06   139.5 2606.97
   159.6 2597.48     170 2589.03   182.5 2575.64   188.3    2574   262.8    2574
   267.7 2575.38   277.3 2576.59   288.8  2575.3   301.9 2579.03   326.4 2581.03
   394.8 2581.01   438.8 2576.93   453.4 2581.24   482.8 2583.64   497.4 2591.31
   534.6 2616.03   544.3 2627.66   551.2 2638.43   562.5 2644.66   597.9 2673.89
#Mann= 3 ,0,0
       0      .1       0   182.5    .045       0   267.7      .1       0
Bank Sta=182.5,267.7
XS Rating Curve= 0 ,0
Exp/Cntr(USF)=0,0
Exp/Cntr=0.3,0.1

Type RM Length L Ch R = 1 ,14241   ,172.1,206,235.5
XS GIS Cut Line= 4
2219502.20118884526875.7575129812219580.28892175527032.005698482
2219809.24517314527175.1975250042219903.07875538527307.442203224
#Sta/Elev= 30
       0 2630.22    64.2 2600.73   104.4 2590.52   117.9 2580.91   135.7 2574.65
   176.9 2577.12     190 2574.14     290 2572.61   294.4 2574.23   303.2 2579.84
   326.4 2577.65   350.4  2579.7   390.2 2579.06   404.7 2581.64     457 2581.56
   476.6  2594.9   491.3 2610.03   502.8 2615.76   505.6 2618.93   510.9 2632.19
   515.8 2635.88   520.7 2634.67   525.8 2627.94   535.4 2621.98   540.3 2622.07
   574.7 2631.97   581.1 2636.09   588.8 2644.58   604.1  2651.3   606.9  2656.4
#Mann= 3 ,-1,0
       0      .1       0     190    .045       0   294.4      .1       0
Bank Sta=190,294.4
XS Rating Curve= 0 ,0
Exp/Cntr(USF)=0,0
Exp/Cntr=0.3,0.1

Type RM Length L Ch R = 1 ,14035   ,381.8,381.9,382.8
XS GIS Cut Line= 2
2219351.40424129 526924.037349022219609.81272132527421.946371506
#Sta/Elev= 30
       0 2635.71    23.8 2623.64    41.8 2617.37    68.9 2603.95    91.4 2595.12
   118.5  2587.8     123 2584.72     132 2575.48   137.9 2573.98   173.5 2575.32
   185.4  2577.5   226.9 2578.58   258.2 2574.51   283.3 2577.05   292.2 2572.44
   298.7 2569.58   334.8 2569.42   366.3 2569.44   375.1 2572.59   387.1  2578.1
     396 2580.41   415.9 2579.96   424.9 2583.52   438.4 2594.41   443.5 2602.99
   447.4 2615.08   465.5 2635.29   528.6 2674.03   537.6 2681.16     561 2695.81
#Mann= 5 ,-1,0
       0      .1       0     132     .04       0   173.5      .1       0
   292.2    .045       0   375.1      .1       0
Bank Sta=292.2,375.1
XS Rating Curve= 0 ,0
Exp/Cntr(USF)=0,0
Exp/Cntr=0.3,0.1

Type RM Length L Ch R = 1 ,13653   ,362.1,353.5,346.2
XS GIS Cut Line= 2
2218997.19554428527067.7376744972219240.47767426527536.654526053
#Sta/Elev= 30
       0 2666.54    21.1 2653.52    37.7 2640.26    49.9 2633.81    64.7 2622.02
      76  2616.5    91.7 2602.64   123.3 2580.93   127.9 2578.87   145.8 2577.47
   163.9 2577.79   168.4 2575.95   174.3 2569.88   177.4 2568.22     208 2568.31
     211 2569.77   217.9 2574.66   228.8 2576.89   285.1 2576.25     299 2574.07
   305.4  2570.9   310.5 2568.28   371.2 2568.22   377.1 2571.09   389.2 2578.05
   416.2 2578.63   427.6 2586.15   442.4 2599.35   463.2 2611.96   528.3 2642.09
#Mann= 5 ,-1,0
       0      .1       0   174.3     .04       0     211      .1       0
   305.4    .045       0   377.1      .1       0
Bank Sta=305.4,377.1
XS Rating Curve= 0 ,0
Exp/Cntr(USF)=0,0
Exp/Cntr=0.3,0.1

Type RM Length L Ch R = 1 ,13299   ,348.9,331.9,313
XS GIS Cut Line= 3
2218593.82620961527356.3988546212218791.72928944527467.325421656
2218987.11131092527745.902368414
#Sta/Elev= 30
       0 2720.28     7.3 2717.02    16.4 2709.65    25.8 2705.63    42.5 2690.83
    53.1 2674.96    55.2 2673.17    80.6 2657.48    94.4 2646.29   116.9 2631.09
     154 2600.14   163.2 2584.95   172.7  2578.3   186.1 2574.12   222.8 2574.74
   234.3 2572.47   253.6  2572.7   274.5 2570.05   282.9 2567.76   297.3 2567.69
   389.3 2567.73   396.2 2569.85   409.4 2574.97   420.9 2576.77   443.9 2574.79
   449.6 2575.62     487 2592.63   495.6 2594.69   521.4 2608.29   567.1  2625.5
#Mann= 3 ,-1,0
       0      .1       0   274.5    .045       0   396.2      .1       0
#XS Ineff= 2 , 0
                          423.89         2590.75
Permanent Ineff=
       F       F
Bank Sta=274.5,396.2
XS Rating Curve= 0 ,0
Exp/Cntr(USF)=0,0
Exp/Cntr=0.3,0.1

Type RM Length L Ch R = 1 ,12968   ,363.2,346.2,331.5
XS GIS Cut Line= 2
2218409.78895067527627.4126263542218837.10833959527938.763331555
#Sta/Elev= 30
       0 2678.95     7.9 2673.06    12.9  2671.2    22.7 2664.66    32.6 2660.61
    54.5 2644.83    82.1 2630.61    94.6 2621.59   131.8 2599.14   141.5 2591.17
   146.5  2589.2   159.2 2580.74   186.2 2567.87     212 2564.79   220.4 2563.37
   266.4 2563.41   272.1 2565.09   280.1 2567.61   326.5 2575.28   352.3 2571.43
   393.9  2570.3   408.8 2567.34   429.6 2567.87   435.3 2571.06   451.3 2586.16
   455.3 2588.74   464.9 2592.82   489.7  2606.8   517.7 2618.05   528.7 2625.45
#Mann= 3 ,0,0
       0      .1       0     212    .045       0   272.1      .1       0
#XS Ineff= 2 , 0
                          329.24         2587.29
Permanent Ineff=
       F       F
Bank Sta=212,272.1
XS Rating Curve= 0 ,0
Exp/Cntr(USF)=0,0
Exp/Cntr=0.3,0.1

Type RM Length L Ch R = 1 ,12621   ,297.9,295,293.8
XS GIS Cut Line= 3
2218208.10428333527989.184498389 2218520.7155177528101.371594594
2218700.97118913528223.642924167
#Sta/Elev= 30
       0 2627.53    18.8 2619.46    34.1 2611.68    59.5    2603   119.4 2579.46
   134.5 2575.24   161.6 2569.88   184.6  2571.6   187.1 2570.99   191.3 2565.47
   195.6 2563.08   200.2    2563   276.3 2563.04  283.38 2565.24   297.2 2568.13
   327.3  2572.4   336.3 2572.05   355.6 2567.56   377.7 2567.71   389.2 2571.08
   397.8  2579.3   406.5 2589.47   418.5 2600.98   435.3 2612.07     462  2631.5
   476.5 2639.74   495.8 2655.54   505.5 2661.13     520  2672.6   549.9 2688.77
#Mann= 3 ,0,0
       0      .1       0   191.3    .045       0  283.38      .1       0
#XS Ineff= 2 , 0
          181.52  2579.7  329.92         2584.45
Permanent Ineff=
       F       F
Bank Sta=191.3,283.38
XS Rating Curve= 0 ,0
Exp/Cntr(USF)=0,0
Exp/Cntr=0.3,0.1

Type RM Length L Ch R = 1 ,12326   ,254.1,237.5,232.9
XS GIS Cut Line= 3
2217998.85644097528236.2482158752218418.61265486 528376.16695384
2218578.69985956528407.680183111
#Sta/Elev= 30
       0 2619.31    15.6 2613.82    73.1 2597.85   106.8 2587.33   172.5 2571.15
   182.7 2570.25   245.9  2573.4   271.2 2573.12   275.5  2572.5   279.7 2570.02
   283.9 2564.59   289.5  2562.4   393.5 2562.25   397.1 2564.53   401.9 2567.22
   418.8 2566.09   425.5    2569   435.7 2571.43   448.1 2571.16   452.2 2571.81
   460.4  2579.9   464.4 2582.41   472.6 2584.09     493 2594.78   517.4  2604.2
     546 2617.66   554.1 2619.96   566.4 2626.75   578.6 2632.33   605.6 2640.97
#Mann= 3 ,-1,0
       0      .1       0   283.9    .045       0   397.1      .1       0
#XS Ineff= 2 , 0
          266.99 2579.85
Permanent Ineff=
       F       F
Bank Sta=283.9,397.1
XS Rating Curve= 0 ,0
Exp/Cntr(USF)=0,0
Exp/Cntr=0.3,0.1

Type RM Length L Ch R = 1 ,12089   ,158.1,152,148.5
XS GIS Cut Line= 3
2217930.78786574528497.1777542412218384.57836725528604.322733764
2218579.96038873528533.733100196
#Sta/Elev= 30
       0    2634    46.6 2603.66    91.8 2583.39   108.3 2577.65   140.8 2570.17
   210.6 2568.87   239.8 2570.01     244 2569.26   252.1 2559.58   256.2 2559.25
   264.5 2560.17   268.6 2563.26   280.9 2564.75   317.9 2564.47   346.7 2561.91
   354.9 2559.32   400.1 2559.32   404.2 2559.79  405.85 2562.01   412.4 2571.92
   416.5 2575.22   445.3 2573.38   453.8 2569.98   470.1 2571.08   478.6 2569.27
   482.9 2570.05   508.4 2591.94   525.4 2592.71     584  2600.3     674 2617.26
#Mann= 3 ,0,0
       0      .1       0   346.7    .045       0  405.85      .1       0
#XS Ineff= 2 , 0
          233.86 2578.04  420.39         2581.88
Permanent Ineff=
       F       F
Bank Sta=346.7,405.85
XS Rating Curve= 0 ,0
Exp/Cntr(USF)=0,0
Exp/Cntr=0.3,0.1

Type RM Length L Ch R = 1 ,11937   ,319.1,236.4,177
XS GIS Cut Line= 5
2217890.45093228528634.575433864 2218187.9358166 528717.77035914
2218312.72820451528736.6782967032218428.69688823528706.425596603
2218556.01033449528595.499029568
#Sta/Elev= 30
       0 2649.45    18.4  2631.6    26.7 2619.05    51.6 2605.04    97.3 2574.25
   138.9 2573.69   191.8 2570.04   214.5 2572.68   243.7 2570.78     251 2569.43
   263.5  2559.6   267.6 2559.19   313.2 2565.54  330.97  2561.6   337.5 2559.19
   398.1 2559.27  401.32 2561.36   406.2 2565.79   426.5 2572.62   440.8 2573.45
   451.1 2570.96   471.7 2581.72   484.2 2577.91   500.7 2576.73   517.2 2570.44
     564 2568.34   586.1 2586.17   589.5 2587.37   672.6 2595.08   723.8 2605.27
#Mann= 3 ,0,0
       0      .1       0  330.97    .045       0  401.32      .1       0
Bank Sta=330.97,401.32
XS Rating Curve= 0 ,0
Exp/Cntr(USF)=0,0
Exp/Cntr=0.3,0.1

Type RM Length L Ch R = 1 ,11700   ,363.9,285.4,230
XS GIS Cut Line= 3
2218084.57242459529142.5686897172218477.85752589528788.359992708
2218574.91827205528608.104321276
#Sta/Elev= 30
       0 2708.35      14 2700.51    26.4 2695.82    48.9 2682.17    61.8 2670.05
    73.8 2651.75    85.7 2637.52   139.5 2603.45   144.8  2598.6   157.5 2578.18
   170.6 2566.57   182.5 2558.99   187.4 2558.22   351.9 2558.89   366.1 2564.96
   372.7 2570.31   380.2 2572.38   456.7  2571.3   473.2 2568.04   489.3 2572.92
   521.8 2567.92   532.9 2569.02   546.5 2567.68   551.1 2569.34   559.9 2576.34
   564.7  2577.8   605.6 2579.25   645.6 2585.29   719.2 2603.62     734 2605.39
#Mann= 3 ,0,0
       0      .1       0   182.5    .045       0   351.9      .1       0
Bank Sta=182.5,351.9
XS Rating Curve= 0 ,0
Exp/Cntr(USF)=0,0
Exp/Cntr=0.3,0.1

Type RM Length L Ch R = 1 ,11415   ,363,365.5,367.3
XS GIS Cut Line= 2
2218548.44715946529240.8899650432218588.78409293528644.659667231
#Sta/Elev= 30
       0 2658.76    15.7 2648.75    23.8 2638.41    27.8  2634.5    59.8 2616.51
    79.9 2607.03    91.9 2603.98     120 2594.12     132 2587.37     136 2583.99
     144 2571.56     148 2567.37  162.72 2556.11   168.1 2553.78   228.2 2553.75
     236 2556.18   264.3 2557.75   280.4 2564.43   284.4 2565.06   328.5 2562.37
   344.5 2567.27   372.6 2566.49   384.6 2568.03   400.6 2566.66   416.3 2572.31
   436.7 2575.44   511.7  2576.9   528.9 2579.19     549 2583.92   597.6 2600.95
#Mann= 3 ,-1,0
       0      .1       0  162.72    .045       0     236      .1       0
#XS Ineff= 2 , 0
                          289.69         2573.47
Permanent Ineff=
       F       F
Bank Sta=162.72,236
XS Rating Curve= 0 ,0
Exp/Cntr(USF)=0,0
Exp/Cntr=0.3,0.1

Type RM Length L Ch R = 1 ,11049   ,207.4,208.9,210.3
XS GIS Cut Line= 3
2218902.65585647529281.2268985112218942.99278994528894.244443059
2218924.08485237528667.349192306
#Sta/Elev= 30
       0  2627.4    16.1 2619.26    48.3 2599.15    68.4 2590.13   108.6 2566.68
   120.7 2564.76   156.9 2565.79   160.9 2563.45   164.9 2559.05   176.2 2553.28
     181 2551.03     185 2550.97   253.4 2550.99     260 2553.56   265.5 2555.23
   293.6 2558.45   321.8  2559.6     354 2559.21     370 2556.44   374.1 2556.85
   382.1 2560.29   394.2 2562.42   414.2 2558.81   430.3 2557.77   478.5 2559.81
   490.5 2564.06   566.8 2578.14   578.8 2582.71   597.3 2592.35   616.8 2597.41
#Mann= 3 ,-1,0
       0      .1       0   176.2    .045       0     260      .1       0
#XS Ineff= 2 , 0
                          390.42         2571.16
Permanent Ineff=
       F       F
Bank Sta=176.2,260
XS Rating Curve= 0 ,0
Exp/Cntr(USF)=0,0
Exp/Cntr=0.3,0.1

Type RM Length L Ch R = 1 ,10841   ,317.6,386.8,443.8
XS GIS Cut Line= 4
2219013.58242351529375.766586324 2219121.9879322529169.039802305
2219158.54327815528889.2023263762219237.95661592528744.241471728
#Sta/Elev= 30
       0 2611.04      12 2609.04    31.4 2603.24    43.6 2600.84    83.1 2588.23
   102.3 2579.45   116.4 2571.41   125.3 2567.73   133.9 2565.62   165.5 2562.35
   249.4 2565.25   253.5 2564.49   257.5 2560.36  261.17  2552.6   261.5 2551.47
   265.6 2550.16   354.3 2550.18   362.4 2552.38   382.5 2554.88   406.7 2555.97
   495.5 2556.81   516.9 2560.96   533.9 2558.39     544 2554.56   556.7 2554.86
     567 2557.64   584.1 2571.85   602.3 2580.78   635.6  2589.5   680.9 2607.02
#Mann= 3 ,0,0
       0      .1       0  261.17    .045       0   362.4      .1       0
#XS Ineff= 2 , 0
                          518.99         2567.15
Permanent Ineff=
       F       F
Bank Sta=261.17,362.4
XS Rating Curve= 0 ,0
Exp/Cntr(USF)=0,0
Exp/Cntr=0.3,0.1

Type RM Length L Ch R = 1 ,10454   ,248.9,264.7,284.6
XS GIS Cut Line= 2
2219014.84295268529404.7587572542219648.88912561529172.821389818
#Sta/Elev= 30
       0 2610.73     9.9 2605.46    48.3 2592.88    69.3 2583.39   124.9  2565.7
   138.5 2564.74   239.9 2565.34   329.4 2563.18   350.7 2561.05   363.5 2554.77
   367.7 2553.85   380.5 2557.23   393.3 2557.28     406 2553.91   423.1 2552.57
   429.6 2549.17   435.9    2547     504    2547     509 2548.78     521 2555.42
   538.1 2558.21   546.4 2565.58   568.3 2581.47   572.2 2584.98   580.7 2595.44
   624.4 2634.24   640.3 2645.88   648.8 2649.26   657.3 2656.57   675.1 2669.08
#Mann= 3 ,-1,0
       0      .1       0   429.6    .045       0     509      .1       0
#XS Ineff= 2 , 0
          385.69 2565.85
Permanent Ineff=
       F       F
Bank Sta=429.6,509
XS Rating Curve= 0 ,0
Exp/Cntr(USF)=0,0
Exp/Cntr=0.3,0.1

Type RM Length L Ch R = 1 ,10189   ,257.2,269.5,286.7
XS GIS Cut Line= 2
2219029.96930273529539.6353785352219710.65505499529486.693153359
#Sta/Elev= 30
       0 2598.44    62.4 2587.74   110.5 2572.29   134.6 2568.84   146.6 2568.44
   170.7 2563.51   371.3 2561.61   379.3 2560.24   387.4 2556.03   391.4 2555.15
   415.5 2554.99   427.5 2548.19   431.5 2546.37     451 2546.35   539.8  2546.4
  545.19 2548.15   563.9 2555.37   575.9 2556.65     580 2560.52     584 2567.22
     592 2576.67     596 2587.85   599.9 2600.36     604 2608.34     608 2612.19
   624.1 2620.77   644.1 2636.93   660.2 2647.67   668.2  2655.9   682.7 2667.61
#Mann= 4 ,-1,0
       0      .1       0     410     .05       0   427.5    .045       0
  545.19      .1       0
#XS Ineff= 2 , 0
          412.51 2564.27
Permanent Ineff=
       F       F
Bank Sta=427.5,545.19
XS Rating Curve= 0 ,0
Exp/Cntr(USF)=0,0
Exp/Cntr=0.3,0.1

Type RM Length L Ch R = 1 ,9919    ,338,344.2,351.9
XS GIS Cut Line= 3
2219011.06136516529702.2436415752219626.19960054529790.480683534
2219781.24468855529721.151579138
#Sta/Elev= 30
       0 2599.95    53.1 2595.57   118.3 2583.48   158.7 2579.25   174.9  2576.3
   197.9 2568.55   227.4 2561.93   247.6 2562.44   271.9 2559.41   360.8 2558.19
   405.2 2559.87   425.4 2557.14   453.7 2545.17   457.8 2542.77   461.8 2542.42
   534.5 2542.44   542.6 2545.22   554.7  2549.3   591.1 2553.64   621.4 2554.27
     633 2560.21   658.7 2567.11   680.6 2578.26   689.3 2579.15   693.6 2582.17
   698.1 2588.71   702.6 2592.49   712.8 2596.79   748.1 2608.73   791.3 2616.72
#Mann= 3 ,-1,0
       0      .1       0   453.7    .045       0   542.6      .1       0
Bank Sta=453.7,542.6
XS Rating Curve= 0 ,0
Exp/Cntr(USF)=0,0
Exp/Cntr=0.3,0.1

Type RM Length L Ch R = 1 ,9575    ,404.7,396.2,385.2
XS GIS Cut Line= 3
2219018.62454019529940.4836548662219258.12508265530064.015513609
2219651.41018396 530168.63943479
#Sta/Elev= 30
       0 2574.57    24.2 2570.57    37.8 2571.25    60.3 2568.93    82.8 2569.68
   185.8  2559.2   267.3 2554.61   300.6 2555.54   321.1 2548.82   350.2  2552.7
   370.9 2552.67   375.1 2552.22   387.5 2543.37   391.6 2540.89   470.3 2540.82
   482.7 2541.05   487.9 2543.49   540.6 2550.09   557.2 2549.84   565.5 2555.88
   569.6 2561.34   573.8 2575.03   577.9 2581.27   589.2  2589.6   598.6 2599.16
   614.7 2609.38     640 2622.69   648.3 2629.17   660.7 2635.86   676.4  2646.6
#Mann= 3 ,-1,0
       0      .1       0   387.5    .045       0   487.9      .1       0
#XS Ineff= 2 , 0
          355.72  2560.2
Permanent Ineff=
       F       F
Bank Sta=387.5,487.9
XS Rating Curve= 0 ,0
Exp/Cntr(USF)=0,0
Exp/Cntr=0.3,0.1

Type RM Length L Ch R = 1 ,9179    ,305,298.6,293
XS GIS Cut Line= 3
2218960.64019833530452.258498231 2219502.6677418530512.763898432
2219682.92341323530472.426964965
#Sta/Elev= 30
       0 2607.81      12    2602    92.1 2573.04   112.7 2566.79   140.4 2553.55
   160.5 2550.32   176.6 2545.63   192.7  2544.4   228.9 2547.91   269.2 2547.48
   322.7 2549.45   329.6 2549.03   333.6 2547.44   340.8 2541.59   345.7 2538.91
   434.2 2538.93   442.1 2541.54   462.4 2544.46   474.5 2544.37   498.6 2549.61
   514.9 2548.31   526.8 2550.03   534.8 2554.21   559.2 2570.73   575.6 2579.13
   628.9 2597.28   641.2 2598.88   657.6 2605.94   682.2 2613.59   730.1 2626.14
#Mann= 3 ,-1,0
       0      .1       0   340.8    .045       0   442.1      .1       0
#XS Ineff= 2 , 0
           322.7 2558.89
Permanent Ineff=
       F       F
Bank Sta=340.8,442.1
XS Rating Curve= 0 ,0
Exp/Cntr(USF)=0,0
Exp/Cntr=0.3,0.1

Type RM Length L Ch R = 1 ,8880    ,361.7,317.3,235
XS GIS Cut Line= 4
2219007.70932345530881.8549016022219262.92757533530793.150996987
  2219488.577859530791.5947881342219726.67781349530673.322915313
#Sta/Elev= 30
       0 2696.68    21.7  2685.7    38.6 2672.16    59.8 2659.05      64 2653.34
    72.5 2631.07   101.5 2609.36   114.8 2596.89   131.8 2584.09   198.9 2541.93
   237.6 2545.13   271.4 2542.47   295.4 2543.03   307.2 2539.36   315.1 2537.67
   395.4 2537.63   443.4 2537.63   451.4 2539.29   467.4 2548.48   483.4 2551.13
   517.7 2550.11   531.1 2546.34     549 2548.48   564.2 2547.18   575.8 2557.19
   580.3 2559.19   593.7 2555.09   607.8 2558.01   651.7 2572.71   761.7  2602.6
#Mann= 3 ,-1,0
       0      .1       0   307.2    .045       0   451.4      .1       0
#XS Ineff= 2 , 0
           233.3 2563.42  494.87         2563.42
Permanent Ineff=
       F       F
Bank Sta=307.2,451.4
XS Rating Curve= 0 ,0
Exp/Cntr(USF)=0,0
Exp/Cntr=0.3,0.1

Type RM Length L Ch R = 1 ,8563    ,373.5,352.5,323
XS GIS Cut Line= 3
2219236.47202483531275.5757413872219480.79681473531007.907818688
2219737.57127546530763.583028782
#Sta/Elev= 30
       0 2676.91    15.6 2672.31    76.7  2645.9    88.6 2642.97    95.3 2636.88
   112.3 2629.61     160 2597.53   168.5 2593.34   183.5 2580.08   188.4 2571.06
   195.4 2552.68  205.97 2537.77     209 2535.38   213.2 2535.19   317.4 2535.24
   322.8 2537.76   328.2 2540.58   349.6 2543.89   405.7 2544.31   430.2 2550.04
   482.4 2549.44   499.7 2543.81   508.2 2544.57   522.3 2549.07   573.3 2546.16
   587.9 2554.96   598.7 2553.78   615.5  2555.9   632.1 2562.32   716.8 2584.16
#Mann= 3 ,0,0
       0      .1       0  205.97    .045       0   322.8      .1       0
#XS Ineff= 2 , 0
                          366.42         2555.58
Permanent Ineff=
       F       F
Bank Sta=205.97,322.8
XS Rating Curve= 0 ,0
Exp/Cntr(USF)=0,0
Exp/Cntr=0.3,0.1

Type RM Length L Ch R = 1 ,8211    ,327.1,336.6,347.2
XS GIS Cut Line= 4
2219648.86737085531423.4155824132219743.79611088531177.534583654
2219767.13924367531065.487546245 2219865.1804014530944.103255719
#Sta/Elev= 30
       0 2662.52    16.7 2653.15    19.8 2650.38      29 2636.45    81.6 2597.23
   118.7 2559.38   131.1 2548.83   146.6 2538.96   165.3 2534.91   173.9 2532.47
   207.7 2532.44   229.6 2532.44   235.6 2535.21   251.1 2540.03   272.1 2540.39
   287.9 2532.58   300.7 2532.57   325.2 2538.91   349.7 2538.36     362 2542.88
   370.2 2549.55     379 2551.24   404.6 2550.35   414.4 2545.27   435.9 2544.69
   443.3  2547.2   455.5 2555.96   467.2 2553.23   487.1 2554.47   534.1 2566.77
#Mann= 3 ,-1,0
       0      .1       0   165.3    .045       0   235.6      .1       0
Bank Sta=165.3,235.6
XS Rating Curve= 0 ,0
Exp/Cntr(USF)=0,0
Exp/Cntr=0.3,0.1

Type RM Length L Ch R = 1 ,7874    ,296.3,295.5,295.2
XS GIS Cut Line= 3
 2219888.5235342531589.9299296732220109.50519131531232.001893506
2220224.66464642531171.309748242
#Sta/Elev= 30
       0 2618.94    10.3 2612.48    32.3 2602.87      45 2595.48    57.3 2591.68
    71.4 2583.19    83.1 2573.86    94.9 2570.74   107.8 2561.83   131.1 2549.32
   151.4 2540.18   174.8 2534.41   197.9 2537.85   221.2  2538.3   231.2 2537.51
   247.3 2532.98   256.1 2529.94   314.2 2529.86   320.5 2530.18   325.2 2532.87
   334.6 2541.12   339.3 2543.14   349.1 2542.14     377 2543.42   381.7 2547.05
   389.8 2556.47   392.7 2557.98   419.3 2560.07   483.9 2572.58   550.8 2582.69
#Mann= 3 ,-1,0
       0      .1       0   247.3    .045       0   325.2      .1       0
Bank Sta=247.3,325.2
XS Rating Curve= 0 ,0
Exp/Cntr(USF)=0,0
Exp/Cntr=0.3,0.1

Type RM Length L Ch R = 1 ,7579    ,324,333.5,341.7
XS GIS Cut Line= 3
2220003.68298931 531781.343618582220181.09079854531680.190043141
2220381.84174057531351.829975179
#Sta/Elev= 30
       0 2620.32    37.4 2598.78    51.2  2592.2    83.4 2572.46   111.9 2556.91
   124.9 2550.31   138.7 2546.63   147.9 2545.49   217.4  2546.5   246.5 2542.61
   282.8 2543.08   296.8  2539.3   320.3 2535.71   348.3 2534.25   357.8  2531.2
   362.5  2529.1   367.2 2528.84   442.2 2528.88   446.9 2529.26   450.1 2531.16
   460.9 2538.59   465.6 2540.41     488 2539.59   503.1 2540.98   521.9 2540.68
   531.2 2542.18   539.9 2545.11     550 2550.89   564.1 2562.13   589.1 2566.32
#Mann= 5 ,-1,0
       0      .1       0   357.8    .045       0   450.1      .1       0
  484.22     .12       0  524.22      .1       0
#XS Ineff= 2 , 0
                          469.52         2547.29
Permanent Ineff=
       F       F
Bank Sta=357.8,450.1
XS Rating Curve= 0 ,0
Exp/Cntr(USF)=0,0
Exp/Cntr=0.3,0.1

Type RM Length L Ch R = 1 ,7245    ,199.6,242.6,292.6
XS GIS Cut Line= 5
2220093.94310278531943.1893392822220276.01953857531894.946864842
2220470.54564518531800.0181248152220646.39724556531594.598556232
2220703.97697312 531566.58679688
#Sta/Elev= 30
       0 2626.13    39.6 2608.56    60.2 2597.43    76.8 2584.75    85.1 2580.03
    93.3 2572.19   101.6 2568.87   109.9 2562.68   137.6 2547.35   151.3 2542.04
   198.8  2543.7   241.9 2539.55   277.5    2542   433.5 2542.18   447.7 2540.09
   461.9 2530.31   487.3 2531.36   495.9 2529.05   499.6  2526.8   505.7 2526.09
   561.1 2526.12   566.8 2529.56   573.4 2534.59   585.7 2538.97   619.2 2540.59
     635  2545.8     652 2556.61   690.5  2587.3   713.5 2595.44   739.3 2600.75
#Mann= 3 ,-1,0
       0      .1       0   495.9    .045       0   566.8      .1       0
Bank Sta=495.9,566.8
XS Rating Curve= 0 ,0
Exp/Cntr(USF)=0,0
Exp/Cntr=0.3,0.1

Type RM Length L Ch R = 1 ,7002    ,293.5,283.5,283.8
XS GIS Cut Line= 4
2220201.63665603532017.5683743782220377.53225704531933.759293896
2220594.81505829531919.2737738132220754.15577921 531932.72461389
#Sta/Elev= 30
       0 2576.54    14.2 2570.53      25 2564.21    35.2 2561.48    53.2  2551.1
    69.3 2545.41    82.6 2543.07   122.4 2542.98   153.5 2539.11   193.3 2541.15
   225.6 2540.36   269.3 2541.46   321.6 2540.09   341.8 2535.81   357.8 2534.53
   381.9 2527.21   397.9 2526.21     410 2531.05     426 2527.42     434    2525
   490.2 2524.97   493.4 2527.13   498.3 2532.11   510.3 2538.26   530.4  2538.5
   534.4 2540.18   538.4 2543.15   546.4 2556.44   558.5 2571.89   572.5 2581.56
#Mann= 3 ,-1,0
       0      .1       0     426    .045       0   493.4      .1       0
Bank Sta=426,493.4
XS Rating Curve= 0 ,0
Exp/Cntr(USF)=0,0
Exp/Cntr=0.3,0.1

Type RM Length L Ch R = 1 ,6719    ,317.1,335,352.8
XS GIS Cut Line= 5
2220162.41629231532318.2356728312220402.07245565532223.306932804
2220493.88877797532196.8513823052220626.16653047532193.738964599
2220823.80505479532223.306932804
#Sta/Elev= 30
       0 2582.94    36.3 2564.24    54.6 2560.82   196.3 2558.69   264.1 2553.94
   280.8 2551.91   322.4 2543.03   351.7 2539.15   359.6 2535.71   371.6 2526.81
   378.7 2523.28   387.6 2520.57   435.6 2520.58   445.1 2523.43   456.9 2526.73
   459.6 2528.08   467.6 2535.74   475.6 2538.17   503.8 2535.48     520 2537.12
   532.2 2536.62   536.3 2537.85   544.3 2545.18   568.6 2572.32   588.8 2585.34
     617 2608.76   649.4 2629.89   664.7 2641.29   676.9 2647.87   685.5  2655.7
#Mann= 3 ,-1,0
       0      .1       0   378.7    .045       0   445.1      .1       0
Bank Sta=378.7,445.1
XS Rating Curve= 0 ,0
Exp/Cntr(USF)=0,0
Exp/Cntr=0.3,0.1

Type RM Length L Ch R = 1 ,6384    ,312.2,320.6,329.9
XS GIS Cut Line= 2
2220296.82721658532437.6484567962220672.41605874532581.468977623
#Sta/Elev= 30
       0 2545.44    23.9 2545.45    80.7 2542.25    89.2 2540.96   127.8  2537.7
   140.6 2537.55   166.3    2539   183.5 2537.79   209.2 2532.81   213.5 2531.06
   225.2 2520.99   230.6 2517.93   234.9 2517.56   277.7 2517.56     282 2518.62
   286.3 2520.67   294.8 2522.69   299.1 2524.76   307.7 2532.87     312 2535.06
   321.2 2534.23   329.1 2535.36   332.9 2537.01   342.9 2544.02   359.1 2553.19
   380.5 2574.31   389.4 2594.61   393.4 2599.34   397.6 2606.91   402.2 2613.97
#Mann= 3 ,-1,0
       0      .1       0   225.2    .045       0   286.3      .1       0
Bank Sta=225.2,286.3
XS Rating Curve= 0 ,0
Exp/Cntr(USF)=0,0
Exp/Cntr=0.3,0.1

Type RM Length L Ch R = 1 ,6063    ,315.9,313,309.2
XS GIS Cut Line= 2
2220062.06021319532610.2331840472220534.06990946532904.349778712
#Sta/Elev= 30
       0 2568.92    26.1 2565.27    82.1 2548.58   111.5 2538.38   143.9 2537.37
   151.8    2536   162.7 2537.81   194.7 2539.24   262.1  2536.8   294.7 2533.43
   305.7 2527.14     326 2520.08   332.4 2516.29   337.1 2515.97   410.2 2516.06
   413.1 2516.52   417.2 2519.86   433.4 2531.98   450.2 2534.02   453.7 2535.94
   464.4 2548.82   483.2  2567.9     506  2586.9   516.2 2593.49   520.9 2599.15
   525.6 2602.57   535.1 2606.42   542.6 2611.66   549.2 2613.52   556.1 2617.45
#Mann= 3 ,-1,0
       0      .1       0     326    .045       0   417.2      .1       0
Bank Sta=326,417.2
XS Rating Curve= 0 ,0
Exp/Cntr(USF)=0,0
Exp/Cntr=0.3,0.1

Type RM Length L Ch R = 1 ,5750    ,345.8,345.7,345.7
XS GIS Cut Line= 2
2219900.77046773532901.9778706912220424.96214048533188.978741291
#Sta/Elev= 30
       0 2560.71    26.7 2553.08   113.3  2541.2   131.5  2534.7   186.3 2532.99
   246.5 2527.29   259.3 2528.61   277.5 2525.31   298.2 2528.54   311.3 2526.36
  324.91 2517.68     329  2515.2   336.8 2514.48   400.6 2514.51   409.7 2517.51
   418.9 2521.31     428 2528.73   432.5 2530.58   441.7 2532.97   455.4 2532.64
   458.7 2533.99   479.3 2556.55   505.5 2569.55   510.1 2572.98   514.7 2579.55
   519.2 2583.59   541.2 2598.24   555.9 2609.85   578.5 2622.57   597.6 2631.14
#Mann= 3 ,0,0
       0      .1       0  324.91    .045       0   409.7      .1       0
#XS Ineff= 2 , 0
          295.77 2536.41
Permanent Ineff=
       F       F
Bank Sta=324.91,409.7
XS Rating Curve= 0 ,0
Exp/Cntr(USF)=0,0
Exp/Cntr=0.3,0.1

Type RM Length L Ch R = 1 ,5405    ,283.5,284.9,286.7
XS GIS Cut Line= 3
 2219765.5717105533222.185453592  2220152.192718533433.285267505
2220320.59818753533502.070600129
#Sta/Elev= 30
       0 2570.94    31.3 2560.89    89.6 2555.18   113.2 2545.58   144.2 2526.82
   157.4 2521.32   176.1 2521.75   194.4 2525.55   221.7 2526.98   276.4 2521.57
   290.1 2518.97  296.39 2516.03   301.9 2512.99   307.8 2512.62   376.7 2512.64
   381.2 2513.15  383.65 2515.98   393.2 2528.65   398.5 2531.14   422.2 2530.31
   444.8    2532   479.4 2530.11   492.3 2532.81   509.6 2544.81   518.3 2549.21
   541.6 2557.15   556.6 2558.79   570.1 2562.74   590.7 2574.54   622.4 2587.63
#Mann= 3 ,0,0
       0      .1       0  296.39    .045       0  383.65      .1       0
#XS Ineff= 2 , 0
          212.96 2538.44
Permanent Ineff=
       F       F
Bank Sta=296.39,383.65
XS Rating Curve= 0 ,0
Exp/Cntr(USF)=0,0
Exp/Cntr=0.3,0.1

Type RM Length L Ch R = 1 ,5120    ,304.3,263.8,208
XS GIS Cut Line= 3
2219720.50545809533513.9301402362220040.71304099533698.938965913
2220311.11055544533691.823241848
#Sta/Elev= 30
       0 2570.07    22.7 2560.54    59.7 2548.04    70.5 2547.31    87.4 2542.91
    96.6  2536.3   105.9 2534.58   110.6 2532.05   124.3 2521.36   133.6 2517.42
   151.5 2513.26   160.2    2513   166.4 2510.57   238.4 2510.71   244.5 2513.13
   253.9 2523.88   259.8 2526.28   272.2 2528.38   350.7 2528.56   373.3  2531.3
   393.3 2528.06   453.3 2529.92   477.3  2528.9   495.8  2530.9   513.3 2536.81
   537.3 2549.09   549.3 2556.89   589.3 2576.21   625.4 2590.26   640.3 2594.66
#Mann= 3 ,-1,0
       0      .1       0   160.2    .045       0   244.5      .1       0
Bank Sta=160.2,244.5
XS Rating Curve= 0 ,0
Exp/Cntr(USF)=0,0
Exp/Cntr=0.3,0.1

Type RM Length L Ch R = 1 ,4856    ,164.1,138.7,109
BEGIN DESCRIPTION:
xs 4
END DESCRIPTION:
XS GIS Cut Line= 3
2219637.25104068533985.0779920172219999.93610828533745.601727286
2220272.38374279 533697.01234024
#Sta/Elev= 30
       0 2580.75     8.3 2577.85      28  2576.8    75.4 2567.28    94.6 2566.04
   113.7 2562.37   128.1  2555.1   137.7 2552.73   161.7 2540.74   176.1 2537.67
  207.48 2510.05   210.3 2508.72     248 2508.78   256.1 2510.08   367.8 2523.08
   377.4 2525.88   410.9 2528.88     443  2528.5   459.1  2531.3   467.4 2531.27
   479.6 2528.31   499.9 2525.85   528.3 2529.81   564.9 2529.99   581.1 2528.25
   593.3 2529.35   601.4 2530.69   621.8 2537.61   682.7 2568.35   711.4 2581.14
#Mann= 3 ,0,0
       0      .1       0  207.48    .045       0   256.1      .1       0
Bank Sta=207.48,256.1
XS Rating Curve= 0 ,0
Exp/Cntr(USF)=0,0
Exp/Cntr=0.5,0.3

Type RM Length L Ch R = 1 ,4717    ,35,34.4,33.4
BEGIN DESCRIPTION:
xs 3
END DESCRIPTION:
XS GIS Cut Line= 6
2219841.04006001534331.8850645142219841.04006001534201.630383526
2219863.44946749 534093.785110022219974.09591693533838.878099914
2220011.91179206533749.2404699872220247.21057061533705.822242991
#Sta/Elev= 30
       0  2538.2    38.7 2534.21    70.7 2535.13    86.7 2534.16   106.7 2535.13
   130.3 2540.17   151.1 2538.66   187.9 2530.85   242.2 2533.51   315.2 2530.64
   329.6  2526.8   345.7 2515.17   354.4 2510.35     363 2508.06   423.1 2508.16
   432.8 2510.48   450.4 2515.98   489.6    2519   502.7 2526.39     509 2527.31
   615.6 2529.59     628 2531.39   660.6 2525.97   693.1 2529.55   762.3 2528.94
   774.5 2531.66   790.4 2537.98     807 2547.14   815.2 2549.62   854.8 2569.24
#Mann= 3 ,-1,0
       0      .1       0   354.4    .045       0   432.8      .1       0
#XS Ineff= 2 , 0
             345 2530.06     441         2530.76
Permanent Ineff=
       F       F
Bank Sta=354.4,432.8
XS Rating Curve= 0 ,0
Exp/Cntr(USF)=0,0
Exp/Cntr=0.5,0.3

Type RM Length L Ch R = 1 ,4683    ,259.4,280,305.6
BEGIN DESCRIPTION:
xs 2
END DESCRIPTION:
XS GIS Cut Line= 6
2219874.65417123534340.288592319 2219876.0547592534218.437439137
2219891.46122684534120.3962814042220013.31238002533829.073984141
2220041.32413938533760.4451737282220233.20469094533725.430474538
#Sta/Elev= 30
       0  2528.7    40.2 2528.18   135.3 2529.61   224.6 2528.95   303.6  2527.4
   311.3 2526.55   318.9 2524.14   331.1 2516.04   341.7 2512.36     345 2510.03
   350.3    2508   419.9 2508.03   428.4 2509.86   445.7    2515   461.4 2516.69
   471.7 2520.44   508.4 2527.42     567 2528.41   613.9 2527.92   626.1  2526.9
   650.5 2529.32   662.7 2528.58     695 2530.84   712.5 2528.29   727.8 2528.62
   735.9 2530.14     744 2532.72   760.3 2539.93   792.8 2557.43   806.1 2563.24
#Mann= 3 ,-1,0
       0      .1       0     345    .045       0   428.4      .1       0
#XS Ineff= 2 , 0
             340    2530     434          2530.5
Permanent Ineff=
       F       F
Bank Sta=345,428.4
XS Rating Curve= 0 ,0
Exp/Cntr(USF)=0,0
Exp/Cntr=0.5,0.3

Type RM Length L Ch R = 1 ,4403    ,345,371.9,406.3
BEGIN DESCRIPTION:
xs 1
END DESCRIPTION:
XS GIS Cut Line= 3
2219919.47298619534338.8880043522220258.41527436534068.574526603
2220367.66113583533893.501030651
#Sta/Elev= 30
       0 2525.65    92.8 2524.29   129.8 2520.02   198.1  2515.8   215.8 2509.17
   256.7 2513.37     285 2512.85   294.9 2511.66   314.8 2506.89   318.1 2505.32
   323.5 2504.81     359 2504.81   363.2 2505.44     366 2507.13   374.6 2510.87
   379.5 2513.92   394.5 2531.45     400 2534.94   420.4 2535.86   432.6 2537.43
   451.7  2537.4   457.6 2539.13   474.6  2546.4   494.1 2551.37   535.1 2558.17
   550.7 2561.67   564.1 2566.42   593.1 2579.28   616.7 2587.92   639.9 2593.82
#Mann= 3 ,-1,0
       0      .1       0   314.8    .045       0     366      .1       0
Bank Sta=314.8,366
XS Rating Curve= 0 ,0
Exp/Cntr(USF)=0,0
Exp/Cntr=0.3,0.1

Type RM Length L Ch R = 1 ,4031    ,233.1,224,210.9
XS GIS Cut Line= 2
  2219927.876514534467.7420973722220453.09700185534480.347389081
#Sta/Elev= 30
       0 2522.64      89 2521.71   100.3  2522.2   112.3    2524   128.3 2524.11
   140.3 2523.22   148.3 2520.84   156.3 2519.47   187.4 2519.74   220.4 2517.03
   236.4 2514.97   272.4 2514.56   288.4  2513.4   296.4 2510.52   308.4 2508.39
   318.2  2504.9   328.4 2502.17   368.4 2502.16   380.4 2502.19   384.4 2503.29
  387.492505.184   392.4 2507.86   404.4 2519.81   428.4 2537.42   449.8 2549.31
   464.4 2558.36   486.7 2570.33   494.9 2577.29   512.4 2595.11   525.4 2604.96
#Mann= 3 ,-1,0
       0      .1       0   318.2    .045       0  387.49      .1       0
#XS Ineff= 2 , 0
           271.1 2521.71
Permanent Ineff=
       F       F
Bank Sta=318.2,387.49
XS Rating Curve= 0 ,0
Exp/Cntr(USF)=0,0
Exp/Cntr=0.3,0.1

Type RM Length L Ch R = 1 ,3807    ,267.5,267.6,268.8
XS GIS Cut Line= 2
2219937.68062977534766.0673344732220471.30464543534663.824412838
#Sta/Elev= 30
       0 2527.04    22.9 2524.51    35.1 2521.04   132.9 2520.47   149.9 2522.03
   206.2 2523.19   214.3 2522.25   226.5 2517.99   234.7 2516.43   291.7 2518.61
   317.3 2514.16   320.2  2512.9   328.4 2504.97   332.4 2502.29   336.5 2501.34
   397.6 2501.34   401.7 2501.75   408.6 2505.18   413.9  2508.7     418 2513.46
   426.7 2519.72   430.3 2524.15   434.3 2531.83   438.3 2537.79   447.2 2546.88
   462.8 2557.59   470.9 2565.03   483.1 2570.33   529.2  2602.1   543.3 2610.39
#Mann= 3 ,0,0
       0      .1       0   328.4    .045       0   408.6      .1       0
Bank Sta=328.4,408.6
XS Rating Curve= 0 ,0
Exp/Cntr(USF)=0,0
Exp/Cntr=0.3,0.1

Type RM Length L Ch R = 1 ,3539    ,248.9,260.9,277.7
XS GIS Cut Line= 2
2219981.09885677535025.1761084822220485.31052511534935.538478555
#Sta/Elev= 30
       0 2525.02    15.3  2525.6    39.7 2521.26    47.8 2518.91    68.1  2516.9
    76.3 2517.06    88.4 2519.46    96.6 2518.34     182 2517.81   202.2 2518.62
   222.5 2516.91   247.6 2517.97   299.3    2516   303.8 2514.21   313.1 2504.04
     316 2501.59     320 2500.72   389.1 2500.72   393.1 2501.34   397.2 2504.12
   413.5 2510.12   423.5 2512.26   429.7 2515.73   441.9 2526.72   451.1 2532.84
   454.1  2535.9   462.2 2547.66   470.3 2555.94   478.7 2560.41   512.1 2581.75
#Mann= 3 ,0,0
       0      .1       0   313.1    .045       0   397.2      .1       0
Bank Sta=313.1,397.2
XS Rating Curve= 0 ,0
Exp/Cntr(USF)=0,0
Exp/Cntr=0.3,0.1

Type RM Length L Ch R = 1 ,3278    ,214.7,216.7,220.8
XS GIS Cut Line= 3
2220044.12531531535238.0654795592220172.97940833535211.454308174
2220509.12052056535238.065479559
#Sta/Elev= 30
       0 2524.92    16.4 2523.15    28.6 2523.64    32.7 2522.76    49.1 2515.33
    57.2 2514.01    73.6 2514.14    85.8 2518.22   114.4 2519.65   150.8 2516.53
   170.9 2513.04     211    2515   235.1 2514.28   251.1 2511.23   263.2 2505.13
   266.3 2502.76   271.2 2499.69   343.4 2499.69  349.29 2502.82   355.5 2507.46
   359.5 2511.84   367.5 2523.52   387.6 2542.86   403.6 2550.55   407.6  2551.4
   419.7 2556.51   438.2 2568.16   444.8 2573.44   459.6 2588.48   468.8  2596.8
#Mann= 3 ,0,0
       0      .1       0   266.3    .045       0  349.29      .1       0
Bank Sta=266.3,349.29
XS Rating Curve= 0 ,0
Exp/Cntr(USF)=0,0
Exp/Cntr=0.3,0.1
